--- MillRun.prj (project) ---

Proj Title=MillRun
Current Plan=p01
Default Exp/Contr=0.3,0.1
SI Units
Geom File=g01
Flow File=f01
Plan File=p01
Background Map Layer=Google Hybrid
Y Axis Title=Elevation
X Axis Title(PF)=Main Channel Distance
X Axis Title(XS)=Station
BEGIN DESCRIPTION:
September 2018
Tucker County ABFE Study
US Army Corps of Engineers, Pittsburgh District
NAD 1983 UTM 17N (meters)
END DESCRIPTION:
DSS Export Rating Curves= 0
DSS Export Rating Curve Sorted= 0
DSS Export Volume Flow Curves= 0
DXF OffsetX= 0
DXF OffsetY= 0
DXF ScaleX= 1
DXF ScaleY= 10

--- MillRun.p01 (plan) ---

Plan Title=MillRun_plan
Program Version=5.05
Short Identifier=Plan1_subcritical
Geom File=g01
Flow File=f01
Subcritical Flow
K Sum by GR= 0
Std Step Tol= 0.003
Critical Tol= 0.003
Num of Std Step Trials= 20
Max Error Tol= 0.1
Flow Tol Ratio= 0.001
Split Flow NTrial= 30
Split Flow Tol= 0.006
Split Flow Ratio= 0.02
Log Output Level= 0
Friction Slope Method= 1
Unsteady Friction Slope Method= 2
Unsteady Bridges Friction Slope Method= 1
Parabolic Critical Depth
Global Vel Dist= 0 , 0 , 0
Global Log Level= 0
CheckData=True
Encroach Param=-1 ,0,0, 0
Computation Interval=1MIN
Output Interval=1HOUR
Instantaneous Interval=1HOUR
Mapping Interval=1HOUR
Computation Time Step Use Courant=        0
Computation Time Step Use Time Series=    0
Computation Time Step Count To Double=0
Computation Time Step Max Doubling=0
Computation Time Step Max Halving=0
Computation Time Step Residence Courant=0
Run HTab= 0
Run UNet= 0
Run Sediment= 0
Run PostProcess= 0
Run WQNet= 0
Run RASMapper=-1
UNET Theta= 1
UNET Theta Warmup= 1
UNET ZTol= 0.006
UNET ZSATol= 0.006
UNET MxIter= 20
UNET Max Iter WO Improvement= 0
UNET MaxInSteps= 0
UNET DtIC= 0
UNET DtMin= 0
UNET MaxCRTS= 20
UNET WFStab= 2
UNET SFStab= 1
UNET WFX= 1
UNET SFX= 1
UNET 1D Methodology=Finite Difference
UNET DSS MLevel= 4
UNET Pardiso=0
UNET DZMax Abort= 30
UNET Use Existing IB Tables=-1
UNET Froude Reduction=False
UNET Froude Limit= 0.8
UNET Froude Power= 4
UNET D1 Cores= 0
UNET D2 Coriolis=0
UNET D2 Cores= 0
UNET D2 Theta= 1
UNET D2 Theta Warmup= 1
UNET D2 Z Tol= 0.003
UNET D2 Volume Tol= 0.003
UNET D2 Max Iterations= 20
UNET D2 Equation= 0
UNET D2 RampUpFraction=0.1
UNET D2 TimeSlices= 1
UNET D2 BCVolumeCheck=0
UNET D1D2 MaxIter= 0
UNET D1D2 ZTol=0.003
UNET D1D2 QTol=0.1
UNET D1D2 MinQTol=0.03
Write IC File= 0
Write IC File at Fixed DateTime=0
Write IC File at Sim End=0
Echo Input=False
Echo Parameters=False
Echo Output=False
Write Detailed= 0
HDF Write Warmup=0
HDF Write Time Slices=0
HDF Flush=0
HDF Face Node Velocities=0
HDF Compression= 1
HDF Chunk Size= 1
HDF Spatial Parts= 1
HDF Use Max Rows=0
HDF Fixed Rows= 1
Calibration Method= 0
Calibration Iterations= 20
Calibration Max Change=0.05
Calibration Tolerance=0.2
Calibration Maximum=1.5
Calibration Minimum=0.5
Calibration Optimization Method= 1
WQ AD Non Conservative
WQ ULTIMATE=-1
WQ Max Comp Step=1HOUR
WQ Output Interval=15MIN
WQ Output Selected Increments= 0
WQ Output face flow=0
WQ Output face velocity=0
WQ Output face area=0
WQ Output face dispersion=0
WQ Output cell volume=0
WQ Output cell surface area=0
WQ Output cell continuity=0
WQ Output cumulative cell continuity=0
WQ Output face conc=0
WQ Output face dconc_dx=0
WQ Output face courant=0
WQ Output face peclet=0
WQ Output face adv mass=0
WQ Output face disp mass=0
WQ Output cell mass=0
WQ Output cell source sink temp=0
WQ Output nsm pathways=0
WQ Output nsm derived pathways=0
WQ Output MaxMinRange=-1
WQ Daily Max Min Mean=-1
WQ Daily Range=0
WQ Daily Time=0
WQ Create Restart=0
WQ Fixed Restart=0
WQ System Summary=0
WQ Write To DSS=0
WQ Use Fixed Temperature=0
Sorting and Armoring Iterations= 10
XS Update Threshold= 0.02
Bed Roughness Predictor= 0
Hydraulics Update Threshold= 0.02
Energy Slope Method= 1
Volume Change Method= 1
Sediment Retention Method= 0
XS Weighting Method= 0
Number of US Weighted Cross Sections= 1
Number of DS Weighted Cross Sections= 1
Upstream XS Weight=0
Main XS Weight=1
Downstream XS Weight=0
Number of DS XS's Weighted with US Boundary= 1
Upstream Boundary Weight= 1
Weight of XSs Associated with US Boundary= 0
Number of US XS's Weighted with DS Boundary= 1
Downstream Boundary Weight= 0.5
Weight of XSs Associated with DS Boundary= 0.5
Percentile Method= 0
Sediment Output Level= 4
Mass or Volume Output= 0
Output Increment Type= 1
Profile and TS Output Increment= 1
XS Output Flag= 0
XS Output Increment= 10
Write Gradation File= 0
Read Gradation Hotstart= 0
Write HDF5 File= 1
Write Binary Output= 1
Write DSS Sediment File= 0
SV Curve= 0
Specific Gage Flag= 0

--- MillRun.f01 (steady flow) ---

Flow Title=MillRun_flow
Program Version=5.05
Number of Profiles= 1
Profile Names=PF 1
River Rch & RM=Mill Run (Cheat),1               ,5029.351
   14.64
River Rch & RM=Mill Run (Cheat),1               ,4754.88
 16.5652
River Rch & RM=Mill Run (Cheat),1               ,4023.411
 26.5043
River Rch & RM=Mill Run (Cheat),1               ,2742.766
 28.4582
River Rch & RM=Mill Run (Cheat),1               ,1920.24
 31.4314
River Rch & RM=Mill Run (Cheat),1               ,182.88
 33.8383
Boundary for River Rch & Prof#=Mill Run (Cheat),1               , 1
Up Type= 2
Dn Type= 1
Dn Known WS=480
DSS Import GetInterval= 0
DSS Import GetPeak= 0
DSS Import FillOption= 0

--- MillRun.g01 (geometry) ---

Geom Title=MillRun_geometry
Program Version=5.05

River Reach=Mill Run (Cheat),1
Reach XY= 30
     619854.5323    4331518.6278     619432.3595    4331575.8314
     619267.2592     4331507.238     619123.1933    4331334.9939
      618986.668    4331408.4159     618738.6206    4331464.3754
     618549.8307    4331645.2906     618492.5576    4331799.3386
     618403.2606    4331813.2292     618362.7793    4331879.9043
      618232.604    4331948.9607     618190.5352     4332072.786
     617950.0284    4332327.5802     617881.3689    4332495.0618
     617722.6186    4332504.9837     617696.4248    4332642.3027
     617620.0487    4332697.7902     617633.7184    4332842.3281
     617560.2965    4332900.1728     617470.6025    4332888.3657
     617405.9117    4332930.4346      617335.767    4333153.0896
     617231.3887    4333287.2336     616973.7836    4333495.5721
616827.795204374   4333486.72289616740.888005631  4333529.976055
      616680.355    4333634.2164     616524.5529    4333642.8343
     616460.9505     4333699.183     616321.4041    4333681.7894

Type RM Length L Ch R = 1 ,5029.351,32.87,31.08,30.36
XS GIS Cut Line= 2
619768.6195260044331482.06569371     619818.8339    4331596.4657
#Sta/Elev= 30
       0     653   2.411 652.443   6.334 651.726   15.84 649.723  22.555 647.653
   29.27 645.287  32.627 644.798  35.984 643.375   38.22 642.287  43.666 638.269
  49.414 635.224  52.771 632.923   55.36  631.31  57.666 630.676  59.486 630.311
  62.844 630.294  66.201 630.753  66.999 631.138  69.558 632.472  72.916 634.727
  76.465 636.899   79.63 639.047  85.665 643.438  89.703   646.2   93.06 646.468
  114.71 660.781 119.919 664.648 120.663 664.975 123.277 665.038 124.935 666.173
#Mann= 3 , 0 , 0
       0      .1       0   55.36      .1       0  66.999      .1       0
Bank Sta=55.36,66.999
XS Rating Curve= 0 ,0
Exp/Cntr=0.3,0.1

Type RM Length L Ch R = 1 ,4998.275,27.47,36.1,38.36
XS GIS Cut Line= 4
     619753.8763     4331493.169      619759.168    4331537.4868
     619767.8993    4331551.9331     619789.9656     4331606.067
#Sta/Elev= 30
       0  654.24    2.98  653.36    5.95  652.21    8.93  650.73   17.85   645.4
   20.83  644.76    23.8  643.71   29.76   640.3   32.73  638.31   35.71  636.07
   38.68  634.23   41.66  632.97   44.63  631.99   47.45  631.34   50.26  631.27
   53.07  630.67   55.89  630.24    58.7  630.35   61.51  631.29   64.44  632.99
   70.28  635.83   79.05  640.97   81.97  642.13    84.9   642.9   87.82  644.92
   90.74  647.51   93.66  649.55   111.2  661.23  114.13  661.51  119.97  665.04
#Mann= 3 , 0 , 0
       0      .1       0   53.07      .1       0    58.7      .1       0
Bank Sta=53.07,58.7
XS Rating Curve= 0 ,0
Exp/Cntr=0.3,0.1

Type RM Length L Ch R = 1 ,4962.17 ,26.07,24.41,24.15
XS GIS Cut Line= 4
     619730.1167    4331492.4017     619730.9105    4331543.3606
     619730.2754    4331559.3944     619744.7217     4331621.307
#Sta/Elev= 30
       0  654.02       3  652.77       6   651.3    8.99   649.7   14.99  646.22
   20.99  642.58   23.98   641.6   26.98  640.86   29.98  639.19   38.97  634.44
   41.97  632.88   44.97   631.5   47.97  630.32   50.97  629.32   53.64  628.74
   58.99  628.65   59.35  628.73   61.66  629.19   70.04   631.9   73.07  633.38
   76.09  635.16   79.12  636.79   82.15  638.02   85.18  638.41   94.26  643.85
  106.37  651.29  112.42  655.12  115.45  655.56  118.48  657.03  130.59  664.71
#Mann= 3 , 0 , 0
       0      .1       0   53.64      .1       0   59.35      .1       0
Bank Sta=53.64,59.35
XS Rating Curve= 0 ,0
Exp/Cntr=0.3,0.1

Type RM Length L Ch R = 1 ,4937.757,91.37,91.47,92.35
XS GIS Cut Line= 3
619701.8472020614331497.63091147     619706.1499    4331542.4544
     619707.3118    4331633.5075
#Sta/Elev= 29
       0 650.021   2.023 649.241     8.2 645.787  14.376 642.446  20.553  639.22
  23.642 639.228  29.818 635.947  39.084 630.863  42.172 629.438  45.259 628.255
  48.334 627.221  51.408 626.851  54.483 626.853  57.557 627.199  60.632 628.068
  66.781 630.614   72.93 633.542  79.079 636.756  79.612 636.903  81.646 636.899
  82.648 637.171   84.76 638.347  85.228 638.479 109.824  652.51 112.899 652.515
 122.122 657.744 125.197  659.57 128.271 661.467  136.09 666.516
#Mann= 3 , 0 , 0
       0      .1       0  48.334      .1       0  57.557      .1       0
Bank Sta=48.334,57.557
XS Rating Curve= 0 ,0
Exp/Cntr=0.3,0.1

Type RM Length L Ch R = 1 ,4846.289,24.7,24.7,24.7
XS GIS Cut Line= 3
619618.571457285 4331534.1230604     619617.4505    4331558.9309
     619616.0304    4331644.0908
#Sta/Elev= 28
       0 626.864   1.899 627.073   2.415 627.199   5.492 627.022    8.57 626.066
  11.647 624.869  14.725 623.862  23.957 622.009  27.032 621.519  30.107 621.715
  33.182 621.482  36.256 622.012  39.331 622.987  42.406 624.187  45.481 625.739
  48.555 627.476  54.705 631.237  57.779 631.236  63.929 635.233  76.228   642.9
  85.452 648.813  88.526 648.813  91.601 650.796  94.676 653.175 100.825 658.736
   103.9 661.283 106.975 663.563 110.005 665.699
#Mann= 3 , 0 , 0
       0      .1       0  23.957      .1       0  36.256      .1       0
Bank Sta=23.957,36.256
XS Rating Curve= 0 ,0
Exp/Cntr=0.3,0.1

Type RM Length L Ch R = 1 ,4832    ,47.2,47.2,47.2
XS GIS Cut Line= 4
619608.7417068044331530.25324127619598.2422646224331550.05218938
619595.8423921234331594.44983061619599.4422008724331641.24734434
#Sta/Elev= 29
       0  623.45   3.631 622.965    9.19 622.834  13.111 622.513  14.071 622.318
  16.012 621.716  18.286 621.132   20.56 620.833  22.411 620.329  24.268 620.007
  27.347 619.669  33.504 619.773  36.583  619.75  39.662 620.103  42.741 620.885
  45.819 622.172  48.898 623.664  58.134 628.833  61.213 630.717  64.292 632.711
  67.371 632.705  73.629 636.846  85.872 644.642  95.122 650.828  98.205 650.824
 101.288 653.214 107.455 658.518 110.538 660.904 113.809 662.998
#Mann= 3 , 0 , 0
       0      .1       0  24.268      .1       0  39.662      .1       0
Bank Sta=24.268,39.662
XS Rating Curve= 0 ,0
Exp/Cntr(USF)=0,0
Exp/Cntr=0.3,0.1

Type RM Length L Ch R = 1 ,4806    ,51.2,51.2,51.2
XS GIS Cut Line= 5
619660.4167667964331461.93257894619588.6005822694331532.12884953
619578.3411273374331551.02784546619576.1812420884331585.04603813
619586.9806683334331646.60276773
#Sta/Elev= 30
       0 626.168   4.508 626.149   11.03 625.738  14.368  625.25  19.726 624.945
  23.165 624.376  34.944 623.418  45.155 622.245  47.988 622.204  50.757 621.562
  53.951  621.22  58.858 621.363  75.942 619.458  78.424 619.554  89.136 618.405
 105.439 617.222 112.435 616.861 123.074 617.159 132.051 618.385 135.131 619.066
 138.212 619.036 144.373 621.092 156.704 627.939 166.067 633.901 169.189 633.939
 178.552 640.522  197.28 653.025 200.401 653.069 212.886 660.762 218.512 663.685
#Mann= 3 , 0 , 0
       0      .1       0 105.439      .1       0 123.074      .1       0
Bank Sta=105.439,123.074
XS Rating Curve= 0 ,0
Exp/Cntr(USF)=0,0
Exp/Cntr=0.3,0.1

Type RM Length L Ch R = 1 ,4754.88 ,42.9,42.9,42.9
XS GIS Cut Line= 4
619503.6577704014331518.65801802     619529.9103    4331570.4373
     619534.6847    4331576.0423     619563.7751    4331643.4294
#Sta/Elev= 30
       0 636.154   13.15 630.969  26.938 625.196  30.385 624.976  34.306 623.413
  40.725 621.326  44.172 620.482  54.512 617.681  57.959 616.918  61.981  616.83
  65.917 615.892  68.318 615.867  69.265 615.964  70.657 616.761  72.614 617.981
  75.962 620.663  82.659 625.296  89.356 629.387  92.705 629.744  96.053 632.106
  99.402 634.629 112.665 644.937 116.144 647.066 119.493 648.802 122.841 650.237
  126.19  650.49 128.178 651.327 133.806 654.058 136.235 655.364 138.815  656.93
#Mann= 3 , 0 , 0
       0      .1       0  61.981      .1       0  70.657      .1       0
Bank Sta=61.981,70.657
XS Rating Curve= 0 ,0
Exp/Cntr=0.3,0.1

Type RM Length L Ch R = 1 ,4712    ,19.4,19.4,19.4
XS GIS Cut Line= 5
619496.3010652714331529.35976404619490.9680152744331631.35434524
619494.9678027714331687.35137021619530.2992590044331752.01460143
619581.6298652284331783.34627016
#Sta/Elev= 30
       0 631.759  16.421  624.68    19.5 624.682  31.813 619.603  41.049 616.479
  47.206 613.264  50.284 613.249  53.363 612.507  56.441 612.077  62.598 611.684
  68.755 611.911  71.834 612.077  83.798 611.997  98.758 612.782 102.619 612.622
 158.274 613.247 172.086 613.903 189.602 614.328 200.111 615.059 214.803 615.494
  231.96 616.544 237.426 617.236 241.028  619.22 251.833 623.489 259.037 626.804
 262.638 630.631 278.628 638.998 280.647 640.242 284.249 644.531 292.097  648.24
#Mann= 3 , 0 , 0
       0      .1       0  56.441      .1       0  68.755      .1       0
Bank Sta=56.441,68.755
XS Rating Curve= 0 ,0
Exp/Cntr(USF)=0,0
Exp/Cntr=0.3,0.1

Type RM Length L Ch R = 1 ,4693    ,29.1,29.1,29.1
XS GIS Cut Line= 2
619484.3861190084331531.58887822619459.5474386464331662.80190709
#Sta/Elev= 30
       0 630.547   8.163 627.136  14.421 624.794   17.55 623.465  20.679 623.473
  29.352 619.341  36.323  616.14  39.452 614.501  42.581 612.585   45.71 611.548
  51.968 611.323   55.66 611.589  61.354 612.162  64.483 612.743  67.612 613.552
  70.741 614.519  74.076 615.886  80.127 619.199  83.256 619.177  84.599 619.645
  85.146 619.955  89.005 621.496  92.643 622.499  95.772  623.13  98.901 623.612
 111.416 624.917 114.545  625.11 120.803 625.812 124.062 626.296 133.543 628.079
#Mann= 3 , 0 , 0
       0      .1       0   45.71      .1       0   55.66      .1       0
Bank Sta=45.71,55.66
XS Rating Curve= 0 ,0
Exp/Cntr(USF)=0,0
Exp/Cntr=0.3,0.1

Type RM Length L Ch R = 1 ,4663.44 ,46.38,42.18,40.46
XS GIS Cut Line= 5
     619478.4468    4331505.8458      619454.955    4331566.6138
     619449.4642     4331570.749     619444.6556     4331580.512
     619422.2227    4331655.9971
#Sta/Elev= 30
       0   639.6   11.85  634.89   17.77  633.72   23.69  631.42   29.61  629.33
   32.58  628.07    38.5  625.01   47.38  620.08   50.34  618.86   53.31  618.39
   62.19  613.71   65.15  611.86   67.44  610.82   70.06  609.87   72.02  609.37
   74.75  609.35   79.64  609.73   88.96  610.13   95.02  611.07  101.08  612.57
  104.11  613.83  116.22  620.27  119.25  620.79  122.28  621.81  140.45  631.02
  143.48  632.09  149.54  635.06  152.57  635.37   155.6  636.78  161.66  638.89
#Mann= 3 , 0 , 0
       0      .1       0   70.06      .1       0   79.64      .1       0
Bank Sta=70.06,79.64
XS Rating Curve= 0 ,0
Exp/Cntr=0.3,0.1

Type RM Length L Ch R = 1 ,4621.258,47.74,49.26,49.43
XS GIS Cut Line= 2
     619436.4418    4331499.0163     619379.2256    4331638.9151
#Sta/Elev= 30
       0  637.95   18.14  628.16   27.21  623.58   30.23  623.39   36.28   620.6
   45.34  616.09   51.39  613.35   57.44  611.06   60.46  610.11   63.48  609.28
    66.5  609.21   69.53  608.62   72.55   608.1   75.57  608.25    78.6  609.33
   84.64  612.54   87.67  613.75   90.69  614.62   93.71  615.18   96.73  615.99
   99.76  616.27  102.78  617.34  108.83  619.96  111.85   621.4  126.96  629.32
  129.99  630.73  133.01  630.89  136.03  632.08   145.1  636.85  151.15   639.8
#Mann= 3 , 0 , 0
       0      .1       0   69.53      .1       0    78.6      .1       0
Bank Sta=69.53,78.6
XS Rating Curve= 0 ,0
Exp/Cntr=0.3,0.1

Type RM Length L Ch R = 1 ,4571.997,91.44,91.44,89.7
XS GIS Cut Line= 4
     619392.5673     4331481.482     619367.7754    4331541.4209
     619364.2297    4331546.2731     619332.3745    4331616.4198
#Sta/Elev= 30
       0  638.43   14.74  626.95   17.69  625.05   20.64  623.93   23.59  623.03
   26.54  621.68   29.48  620.11   32.43  619.19   38.33  616.23   44.23  613.72
   50.12   611.4   56.02  609.38   58.97  609.08   61.92  608.27   64.86   607.3
   70.87  604.94   73.84  604.47    76.8  605.14   79.76  607.14   82.73  608.91
   88.65  611.65   91.62  612.72   94.58  613.23   100.5  615.74  103.47  617.18
  127.17  629.94  130.14  630.34   133.1  631.48  139.03  634.72  147.91  639.78
#Mann= 3 , 0 , 0
       0      .1       0   70.87      .1       0    76.8      .1       0
Bank Sta=70.87,76.8
XS Rating Curve= 0 ,0
Exp/Cntr=0.3,0.1

Type RM Length L Ch R = 1 ,4480.56 ,87.92,91.44,94.63
XS GIS Cut Line= 2
     619322.3899    4331439.9107     619250.6749    4331573.9044
#Sta/Elev= 30
       0  629.23    6.08   626.6    9.12  625.46   12.16  624.53    15.2  624.12
   18.24  623.35   24.32  621.31    30.4  618.82   33.44     617   36.47  614.85
   39.51  613.45   45.59  609.15   51.67  607.29   54.71  606.01   63.83  602.79
   66.87  602.03   79.03  599.78   82.07  599.36   87.38  599.64   88.15  599.65
   91.19  600.63  100.31  605.13  103.35  606.49  112.46  609.89  118.54  613.33
  124.62  615.72  127.66  617.23  142.86  625.82  148.94  629.66  151.98  631.26
#Mann= 3 , 0 , 0
       0      .1       0   79.03      .1       0   87.38      .1       0
Bank Sta=79.03,87.38
XS Rating Curve= 0 ,0
Exp/Cntr=0.3,0.1

Type RM Length L Ch R = 1 ,4389.12 ,97.03,91.44,86.85
XS GIS Cut Line= 4
     619313.1921    4331410.0444     619226.0591    4331447.6657
     619219.2542    4331449.9989     619155.7647    4331482.1435
#Sta/Elev= 29
       0  630.89    3.06  628.61   18.37  622.39   21.43  621.21   27.55  618.07
    39.8  613.92   45.92  612.05   48.98  610.33   52.05  609.09   70.42  603.09
   73.48   601.7   85.72  598.32   91.85  596.31   94.91  595.69   97.31  595.63
   102.1  595.97  116.93  597.13  119.89  598.01  122.86  599.38  140.65  609.84
  143.61  612.65  146.58  614.18  149.54  615.34  152.51  616.93   161.4  622.55
  164.37  624.47  167.33  627.36   170.3  629.84  173.26  631.58
#Mann= 3 , 0 , 0
       0      .1       0   91.85      .1       0   102.1      .1       0
Bank Sta=91.85,102.1
XS Rating Curve= 0 ,0
Exp/Cntr=0.3,0.1

Type RM Length L Ch R = 1 ,4297.68 ,33.24,30.7,25.69
XS GIS Cut Line= 3
     619245.5984    4331322.1662      619151.337    4331394.4334
     619125.3376    4331447.0861
#Sta/Elev= 30
       0  630.86    3.05  629.23    6.09  626.98    9.14  625.08   30.46  614.16
    33.5  611.84   36.55  610.87   39.59  609.69   48.73  605.81   57.87  601.71
   60.91  600.49      67  596.92   70.05  595.49   73.09  594.93   79.18   595.4
   91.37  594.88   100.5  594.87  112.69  595.05  115.73  595.29  121.71  597.52
  124.65  598.76  127.58  600.31  139.33  607.39  142.26  608.08   145.2  609.22
  154.01   614.6  159.88   618.8  171.63   627.5  174.56  629.23   177.5  629.73
#Mann= 3 , 0 , 0
       0      .1       0   70.05      .1       0  112.69      .1       0
Bank Sta=70.05,112.69
XS Rating Curve= 0 ,0
Exp/Cntr=0.3,0.1

Type RM Length L Ch R = 1 ,4266.98 ,26.46,25.24,21.57
XS GIS Cut Line= 5
       619221.71    4331293.9859     619168.4625    4331337.3115
     619159.7841    4331355.3164      619144.941    4331368.8896
     619122.6127    4331432.7151
#Sta/Elev= 30
       0  628.49   23.88  615.35   26.86  612.89   29.85  610.89    38.8   606.3
   41.79   605.4   44.77  604.22   47.75  602.76   56.71  598.77   68.65  595.41
    71.5   594.7   74.36  594.23   77.21  594.15   94.38  594.55   97.25  594.72
  108.75  594.92  117.97  595.23  121.04  595.51  124.12     596  127.19  596.22
  133.34  597.92  136.41  598.94  139.48   600.2  142.56  601.83  145.63  603.74
  154.85  609.99  157.92   611.7     161  612.59  164.07  613.73  176.37  621.94
#Mann= 3 , 0 , 0
       0      .1       0   74.36      .1       0   94.38      .1       0
Bank Sta=74.36,94.38
XS Rating Curve= 0 ,0
Exp/Cntr=0.3,0.1

Type RM Length L Ch R = 1 ,4241.746,37.28,35.51,31.98
XS GIS Cut Line= 5
     619147.5365    4331263.6461     619146.7428    4331306.8261
      619142.774    4331326.1937     619137.3099    4331353.8647
     619118.2598    4331429.9854
#Sta/Elev= 30
       0  622.06    2.88  621.69   11.52  615.64    14.4  613.74   20.15  610.34
   28.79   605.7   34.55  604.25   37.43  602.75   40.31  601.45   43.19   600.4
   54.48  596.97   60.13  594.93    68.6  593.74   79.88  593.58    82.7  593.77
   88.34  594.53   91.16  594.75  106.25  594.81  115.31  595.35  118.32  595.82
  121.34  596.68  124.36  597.81  127.38  597.82  136.43  601.75  139.45  603.38
   148.5  609.15  154.54  612.77  160.58   614.5  163.59   616.3  169.63  620.35
#Mann= 3 , 0 , 0
       0      .1       0    68.6      .1       0    82.7      .1       0
Bank Sta=68.6,82.7
XS Rating Curve= 0 ,0
Exp/Cntr=0.3,0.1

Type RM Length L Ch R = 1 ,4206.24 ,94.01,91.55,89.98
XS GIS Cut Line= 3
     619092.2578    4331270.8675     619115.0619    4331386.9628
     619112.1084    4331429.8881
#Sta/Elev= 30
       0  621.16    3.03  620.08     9.1  616.34   21.24  608.56    27.3  604.96
   30.34  603.69   33.37  603.24   39.44  599.72   51.57  592.27   54.61   591.4
   57.64  591.18   60.67  591.18   66.74  591.44   69.77  591.36   75.84  591.52
   78.88   591.7   81.91  592.04   87.98  593.24   91.01  593.53   94.04  594.04
  115.28  599.34  121.39  600.27  124.46  601.42  127.53  602.77  130.61   604.4
  145.97  613.16  149.05  614.42  152.12  615.04  158.27  618.96  161.34   621.1
#Mann= 3 , 0 , 0
       0      .1       0   54.61      .1       0   66.74      .1       0
Bank Sta=54.61,66.74
XS Rating Curve= 0 ,0
Exp/Cntr=0.3,0.1

Type RM Length L Ch R = 1 ,4114.691,70.8,70.8,70.8
XS GIS Cut Line= 3
618983.890750047  4331309.467047     619008.6401    4331351.6216
     619064.8802     4331451.584
#Sta/Elev= 30
       0 605.079   6.634 604.642  10.199 605.178  24.459 603.839  27.212 604.198
  31.901 603.131  38.719 600.929  42.284 600.924  45.849 599.632  49.408 597.977
   59.99 591.379  62.697 590.069  70.573 588.194    74.1 588.071  81.155 586.877
   88.21 586.507  90.311 586.993  91.737 587.376  95.265  589.36  102.32 591.256
 105.847 591.568 110.627 593.242 125.394 600.642 131.664 604.768 134.066 605.981
 137.594 606.504 149.003 612.414 158.758  617.77 162.286 620.568  163.58 621.404
#Mann= 3 , 0 , 0
       0      .1       0  81.155      .1       0  90.311      .1       0
Bank Sta=81.155,90.311
XS Rating Curve= 0 ,0
Exp/Cntr=0.3,0.1

Type RM Length L Ch R = 1 ,4044    ,20.4,20.4,20.4
XS GIS Cut Line= 4
618955.2142330194331324.23989432618959.5340035174331399.83587804
618968.7135158254331426.83444365619020.0107904874331482.45148881
#Sta/Elev= 30
       0 594.559   3.251 594.169    6.33 593.278  14.612   591.5  19.333 591.015
  24.806 590.138  27.885 589.981  40.202 587.437   49.44 585.827  52.519 585.357
  55.598 585.327  67.916 583.977  77.276 582.662  83.726  582.53   90.22 582.654
  91.815 583.106  93.467 583.606 103.209 587.348 115.459 591.042 119.642 591.412
 123.543 592.935 128.006 595.228 150.444 604.859   153.1 606.388 154.979 606.922
 157.282 607.251 162.704 609.747 168.582 612.719 177.651 617.794 179.897 619.619
#Mann= 3 , 0 , 0
       0      .1       0  77.276      .1       0  91.815      .1       0
Bank Sta=77.276,91.815
XS Rating Curve= 0 ,0
Exp/Cntr(USF)=0,0
Exp/Cntr=0.3,0.1

Type RM Length L Ch R = 1 ,4023.411,84.86,91.49,94.99
XS GIS Cut Line= 3
618885.7638598764331346.86426925     618940.4786    4331411.4676
     619014.8738    4331490.9012
#Sta/Elev= 30
       0 624.132   6.834  618.81  10.863  615.22  12.802 614.169  15.091 614.457
  25.889 606.299  31.006   603.5  39.064 600.127  47.121 598.164   51.15 598.394
  55.179 597.231  62.971 594.457  76.929  588.03  79.351 586.648  83.379 583.557
  87.533 582.489  89.134 581.833  91.309 581.469   95.34 582.762 117.827 588.493
  121.23 589.782 125.442 590.444 128.284 591.525 144.811 598.445 149.308 600.955
 154.926 603.332 159.138 603.927 171.795 609.365 192.834 621.497 193.492 621.623
#Mann= 3 , 0 , 0
       0      .1       0  87.533      .1       0   95.34      .1       0
Bank Sta=87.533,95.34
XS Rating Curve= 0 ,0
Exp/Cntr=0.3,0.1

Type RM Length L Ch R = 1 ,3931.92 ,95.7,91.44,91.88
XS GIS Cut Line= 3
     618846.3374    4331342.6062     618858.6284    4331437.5511
     618875.1736    4331518.6825
#Sta/Elev= 30
       0  620.94   17.95  605.75   20.94  604.81   23.93  603.41   32.91  596.36
    35.9   594.4   38.89  592.98   47.87  589.58   50.86  588.82   53.85  588.48
    71.8  581.23   77.79  579.78   83.77  579.21   86.76  578.56   89.75  578.15
   92.75  578.14   95.74  578.49     108  580.57  111.07  580.82  114.14  582.26
  120.27  586.94  123.34  588.83  132.54  593.34  138.67  597.01   144.8  599.19
     154   605.8  166.27  615.51  169.34  617.12   172.4  617.75  178.54  621.27
#Mann= 3 , 0 , 0
       0      .1       0   86.76      .1       0   95.74      .1       0
Bank Sta=86.76,95.74
XS Rating Curve= 0 ,0
Exp/Cntr=0.3,0.1

Type RM Length L Ch R = 1 ,3840.48 ,95.56,91.44,87.03
XS GIS Cut Line= 4
     618724.3607    4331398.0322     618767.7245    4331445.8702
     618770.0185    4331461.2685     618798.1796    4331540.1138
#Sta/Elev= 30
       0  612.62    2.93   609.3    5.87  606.36   11.74  601.71   17.61  598.26
   20.54  595.37   26.41  590.11   29.35  586.85   32.28  584.63   41.09  580.35
   49.89  576.99   52.83  576.86   61.63  574.85   64.57   574.5   69.76  574.12
   72.35   574.2   74.95  574.78   80.14  576.23   86.12  576.96   95.09  579.17
  104.06  582.27  110.04  585.26  116.02  586.85  127.98  592.56  142.93  600.17
  145.92  601.26  148.91  603.23   151.9  605.61  157.88  609.23  163.86  613.31
#Mann= 3 , 0 , 0
       0      .1       0   64.57      .1       0   74.95      .1       0
Bank Sta=64.57,74.95
XS Rating Curve= 0 ,0
Exp/Cntr=0.3,0.1

Type RM Length L Ch R = 1 ,3749.04 ,81.86,91.44,101.07
XS GIS Cut Line= 4
     618624.1099    4331463.9136     618678.4987    4331504.6496
     618748.5037    4331526.3755     618782.8602    4331557.5763
#Sta/Elev= 30
       0  611.15   11.82  604.88   17.73  601.39   23.64  598.26   29.54  597.25
   38.41  592.79   59.09  583.52      65  579.57   67.95  578.33   71.01  577.85
   74.06  577.79   83.22  575.72   86.28  574.36   95.44  571.36   98.49  570.77
  101.55  570.66   104.6  571.43  113.76   573.1  122.93  575.31  129.03  578.83
   138.2  583.37  141.25  584.27  144.15  585.42  149.95  589.46  167.36  597.66
  170.26  599.35  173.16  602.09  178.96  605.96  184.76  608.75  187.66  610.42
#Mann= 3 , 0 , 0
       0      .1       0   95.44      .1       0   104.6      .1       0
Bank Sta=95.44,104.6
XS Rating Curve= 0 ,0
Exp/Cntr=0.3,0.1

Type RM Length L Ch R = 1 ,3657.6  ,29.3,29.3,29.3
XS GIS Cut Line= 4
     618599.5036    4331473.4386      618634.716    4331529.2432
     618650.4932    4331614.0451       618681.26    4331656.0015
#Sta/Elev= 30
       0  603.91       6  599.79      12  596.15      15   595.6      18  594.64
   23.99  591.67   44.99  582.85   47.99  582.54   50.99  581.64   59.99  577.51
   62.99  575.77   65.99   574.8   74.91  572.49   80.86  571.75   86.81  570.37
  105.07  566.89  107.63  566.58  113.55  566.83   122.5  568.64  125.47  569.58
   134.4  573.39  140.34  574.71  146.29  576.85  164.48   582.4  170.61  584.65
  182.85     591  195.09  597.88  198.15  600.16  201.21  602.83  204.27  603.72
#Mann= 3 , 0 , 0
       0      .1       0  105.07      .1       0  113.55      .1       0
Bank Sta=105.07,113.55
XS Rating Curve= 0 ,0
Exp/Cntr=0.3,0.1

Type RM Length L Ch R = 1 ,3628    ,62.3,62.3,62.3
XS GIS Cut Line= 4
618580.4741423284331474.35191912618604.7728513794331545.62813234
618623.6718473074331610.42468981618662.0098104764331662.26193578
#Sta/Elev= 30
       0 597.814   7.234 595.242   13.73 591.849  16.978 592.084  26.722 586.163
  33.129 582.759  40.462 579.964  42.962 578.558   46.21 578.837  52.706 575.808
   62.45 572.286  67.107 571.568   75.44 569.255  78.642 569.062  88.249  566.96
  92.579 566.426 110.666 565.294 113.868 565.091 118.978 565.399 133.083 567.639
 136.285 567.787 139.487 569.554 154.651 574.453 187.622 583.557 192.376 585.741
 196.703 588.271 200.024 591.241 201.873 592.328 203.847 592.922 207.275 595.003
#Mann= 3 , 0 , 0
       0      .1       0 110.666      .1       0 118.978      .1       0
Bank Sta=110.666,118.978
XS Rating Curve= 0 ,0
Exp/Cntr(USF)=0,0
Exp/Cntr=0.3,0.1

Type RM Length L Ch R = 1 ,3565.997,97.8,91.28,88.83
XS GIS Cut Line= 2
     618517.7472    4331567.8951     618647.9225    4331699.6579
#Sta/Elev= 30
       0  602.59    9.11  597.69   15.18  593.73   21.25  588.61   24.29  587.57
   27.33     585    33.4  578.79   36.44   575.2   39.47  572.16   42.51  570.75
   57.69  565.61   60.73  564.77   72.87  562.49   75.91  562.06   79.22  562.33
   81.98  563.21   91.09  568.46   94.13  569.75   100.2   570.2  118.42  570.46
  127.53  571.89   133.6  573.29  136.64  574.41  139.68  576.12  148.78  579.83
  160.93  585.57  170.04  591.95  173.08  593.76  176.11  594.92  185.22  600.86
#Mann= 3 , 0 , 0
       0      .1       0   72.87      .1       0   79.22      .1       0
Bank Sta=72.87,79.22
XS Rating Curve= 0 ,0
Exp/Cntr=0.3,0.1

Type RM Length L Ch R = 1 ,3474.72 ,88.36,91.44,93.53
XS GIS Cut Line= 4
     618413.7658    4331648.8577     618482.2716    4331687.5727
     618564.0747    4331708.0235     618620.1412    4331739.3454
#Sta/Elev= 30
       0  603.05    3.03  601.14   15.13  595.71   21.19  594.15   24.21  592.39
   42.37  584.38    45.4  582.79   66.58  574.45   72.64  570.14   78.69  565.33
    81.7  563.77   90.73  561.77   108.8  559.56  117.84     559  120.85  559.69
  129.88   565.3  132.89  565.82  144.94  566.58  153.97  566.86     160  567.93
  166.07   569.8  169.13   571.7  187.47  581.17  190.53  582.97  193.59  585.61
  196.65   587.2  202.77  589.42  211.94   594.4     215  597.07  227.23  603.39
#Mann= 3 , 0 , 0
       0      .1       0   108.8      .1       0  120.85      .1       0
Bank Sta=108.8,120.85
XS Rating Curve= 0 ,0
Exp/Cntr=0.3,0.1

Type RM Length L Ch R = 1 ,3383.28 ,81.39,91.47,91.37
XS GIS Cut Line= 4
     618362.2513    4331669.7334     618458.1647    4331768.5017
     618492.1599    4331781.4386     618560.3074    4331820.6235
#Sta/Elev= 30
       0  602.31    9.18     599    15.3  596.04   30.59  590.47   33.65  589.57
   36.71   589.2   45.89  585.49   58.13  581.75   64.25   579.6   70.37  576.95
   76.49  575.79   88.72  571.69   91.78  570.27    97.9  568.29  104.02  566.74
  110.14     566  116.26  564.43  140.71   559.5  164.96  556.99   180.1  556.58
  183.12  556.77  186.14  558.18  195.21  566.49  201.26  575.39  207.31  582.36
  222.42  589.04  228.47  592.56  243.59   598.8  249.64  601.94  252.66  602.79
#Mann= 3 , 0 , 0
       0      .1       0  164.96      .1       0  183.12      .1       0
Bank Sta=164.96,183.12
XS Rating Curve= 0 ,0
Exp/Cntr=0.3,0.1

Type RM Length L Ch R = 1 ,3291.81 ,99.37,91.41,78.36
XS GIS Cut Line= 2
     618371.7763     4331693.546     618466.2327    4331926.9089
#Sta/Elev= 30
       0  593.04    3.07  592.68    9.21  590.71    30.7  582.78   36.84  581.15
   39.91  579.45   55.26  573.28    61.4  571.76   67.54  570.91   82.89  567.01
   98.25  564.39   113.6  559.17  119.74  556.11  122.81  555.02  132.02  555.42
  138.16  555.73  147.37   556.9  165.79  560.78     175  560.42  178.07   560.6
  181.14  561.52  184.21  562.96  190.35  564.83  199.56  569.98  208.77  576.27
  214.91  579.59  217.98  580.19  245.61  592.74  248.68  593.53  251.75  594.82
#Mann= 3 , 0 , 0
       0      .1       0  122.81      .1       0  132.02      .1       0
Bank Sta=122.81,132.02
XS Rating Curve= 0 ,0
Exp/Cntr=0.3,0.1

Type RM Length L Ch R = 1 ,3200.4  ,89.66,91.54,94.84
XS GIS Cut Line= 2
     618292.2839    4331819.2282      618438.351    4331932.5042
#Sta/Elev= 30
       0  583.37    6.06  579.37    9.09  577.96   12.12  577.46   15.15  576.04
   24.24  571.52   27.27   569.2    30.3  567.48   33.33  566.35   45.45  563.13
   51.51  561.14   54.54  560.77    69.7  556.64   75.76   554.4   87.88  553.32
   93.94  552.85   96.97  552.99     100  553.75  106.06  555.76  118.18  557.09
  133.33  560.17  136.36  560.45  139.39  561.36  142.42  563.07  145.45  565.35
  163.63  574.37  169.69  578.38  175.75  581.23  181.81  583.24  184.84  584.68
#Mann= 3 , 0 , 0
       0      .1       0   87.88      .1       0   96.97      .1       0
Bank Sta=87.88,96.97
XS Rating Curve= 0 ,0
Exp/Cntr=0.3,0.1

Type RM Length L Ch R = 1 ,3108.864,94.02,91.4,79.73
XS GIS Cut Line= 2
      618241.601    4331847.5338     618355.9435    4332020.0494
#Sta/Elev= 30
       0  584.97    9.13     580   12.17  577.98   15.22  576.34   18.26  575.74
   42.61  565.23    48.7   561.6   51.74  560.91   54.79  559.41   57.83  557.67
   63.92  553.52   66.96  552.32      70  551.72   73.05  551.19   76.09  551.31
   79.13  551.94    97.4  554.23  109.57   554.8  136.96  555.19  152.18  555.71
  155.23   555.9  158.27  556.64  164.36   560.3  170.44  565.48  179.58  571.74
  182.62  572.71  185.66  574.19  191.75  578.01  203.92  585.06  206.97  586.27
#Mann= 3 , 0 , 0
       0      .1       0      70      .1       0   79.13      .1       0
Bank Sta=70,79.13
XS Rating Curve= 0 ,0
Exp/Cntr=0.3,0.1

Type RM Length L Ch R = 1 ,3017.459,91.99,91.39,87.16
XS GIS Cut Line= 3
     618146.7477    4331940.3366     618231.0824    4331977.9855
     618330.8981    4332055.4305
#Sta/Elev= 30
       0  585.37   11.92  581.42    14.9  579.82   29.79   574.3   32.77  573.04
   35.75  571.31   38.73  570.22   41.71  569.16   50.65  566.95   53.63   565.5
   65.54  558.01   77.46  548.83   80.44  548.49   83.42  549.03   89.38  550.16
  101.38  551.53  119.43  552.95  143.49  555.27  149.51  557.46  164.55   564.1
  167.56  565.59  170.57  567.96  176.58  571.26  179.59  572.42  188.61  574.69
  191.62  576.15  194.63  578.01  200.65  580.29  209.67  583.12  218.69   585.6
#Mann= 3 , 0 , 0
       0      .1       0   77.46      .1       0   83.42      .1       0
Bank Sta=77.46,83.42
XS Rating Curve= 0 ,0
Exp/Cntr=0.3,0.1

Type RM Length L Ch R = 1 ,2926.065,89.17,91.41,93.33
XS GIS Cut Line= 3
     618095.9476     4332018.918     618150.1475    4332046.1984
     618277.7167    4332084.7993
#Sta/Elev= 30
       0  584.47   12.14  579.41    18.2  575.46   30.34  569.34   33.37  567.59
   39.44  562.39   48.54  556.72   51.58  555.41   57.64  553.82   72.79  551.74
   78.85  550.18   87.94  548.33   97.03   547.2  103.09  545.97  109.03  545.54
  112.17  545.69   115.2  546.37  118.23  548.55  121.26  551.13  133.38  557.94
  136.41  559.82  139.44  562.95  148.52  568.04  157.61  571.38  163.67  574.45
  169.73  576.47  178.81  579.06  184.87  581.58  190.93  584.54  193.96  585.68
#Mann= 3 , 0 , 0
       0      .1       0  103.09      .1       0  112.17      .1       0
Bank Sta=103.09,112.17
XS Rating Curve= 0 ,0
Exp/Cntr=0.3,0.1

Type RM Length L Ch R = 1 ,2834.65 ,93.74,91.88,90.96
XS GIS Cut Line= 3
     618074.5163    4332060.9868     618129.5176    4332118.1781
     618184.8478    4332166.5558
#Sta/Elev= 30
       0  584.79    3.05  583.71     6.1     583    9.16  581.58   12.21  579.48
   15.26  577.75   24.41   573.4   27.47  571.61   33.57  567.62   36.62  565.35
   39.67  562.29   45.78  559.37   57.98  550.64   67.14  545.08   70.19  544.14
    75.4  543.16   82.41  542.77   85.47  543.34   88.53  545.15    91.6  548.63
   94.66  550.79  113.03  562.09   116.1  564.91  119.16  566.06  122.22  567.58
  131.41  573.85  137.53  577.67  140.59  580.11  143.66  581.77  152.84   585.8
#Mann= 3 , 0 , 0
       0      .1       0    75.4      .1       0   85.47      .1       0
Bank Sta=75.4,85.47
XS Rating Curve= 0 ,0
Exp/Cntr=0.3,0.1

Type RM Length L Ch R = 1 ,2742.766,49.8,49.8,49.8
XS GIS Cut Line= 2
      617992.998    4332154.8876     618148.5733     4332220.769
#Sta/Elev= 30
       0  585.56    3.07  583.35   12.29  578.88   18.43  576.48    21.5  574.53
   27.65  571.71   36.86  566.87   39.93  565.14   43.01  562.73   46.08  560.75
   61.44  552.87   64.51  550.38   67.58  548.52   73.72  545.51   82.94     542
   85.11  540.82   86.01  540.33   89.08  540.02   92.15  540.39  101.37   544.3
  122.87  556.45  125.94  558.59  129.02  561.52   141.3  567.77  144.38  569.64
  150.52  575.21  153.59  577.18  159.73  580.78  165.88  583.53  168.95  585.32
#Mann= 3 , 0 , 0
       0      .1       0   85.11      .1       0   92.15      .1       0
Bank Sta=85.11,92.15
XS Rating Curve= 0 ,0
Exp/Cntr=0.3,0.1

Type RM Length L Ch R = 1 ,2693    ,40.5,40.5,40.5
XS GIS Cut Line= 4
618014.0442357954332195.21362096618039.9628587824332225.45201444
618078.3008219514332249.21075218618171.7158589674332293.48839979
#Sta/Elev= 30
       0  563.28  11.115 557.714    17.6 554.772  22.324 551.768   31.36 547.976
  35.409 547.059  48.127 541.609  58.977 539.354  62.594 539.024   66.21  539.08
  67.077 539.404  68.476 539.689  71.543 541.123  73.776 541.592  80.148  542.04
  82.708 543.182  84.929  543.86  86.227  543.98  89.557 545.313  93.404 546.104
   98.79  547.87 105.714 549.058 119.563 550.771 122.115 550.887 126.487 551.729
 131.962 551.875 150.826 554.289 179.536 561.531 186.714 561.947 188.307 562.329
#Mann= 3 , 0 , 0
       0      .1       0  58.977      .1       0  67.077      .1       0
Bank Sta=58.977,67.077
XS Rating Curve= 0 ,0
Exp/Cntr(USF)=0,0
Exp/Cntr=0.3,0.1

Type RM Length L Ch R = 1 ,2652.452,93.6,92.65,90.67
XS GIS Cut Line= 2
     617978.7105    4332178.7002     618073.9607     4332332.688
#Sta/Elev= 30
       0  584.27   15.34   575.9   18.41  573.16   21.48  572.39   30.69  567.71
   46.03  560.77   52.17  557.66   55.24  556.72   76.72  547.11   85.93  542.78
      89  541.72   92.07   540.9   104.7  538.18  107.41  537.75  110.48  537.93
  111.65  538.57  113.55  539.61  116.62  542.54  119.69   543.7  128.89  549.64
  144.24  558.59  147.31  560.48  153.45  564.37  159.58  568.46  162.65  570.57
  165.72  572.97  171.86  578.84  174.93  581.47     178  583.86  181.07  585.97
#Mann= 3 , 0 , 0
       0      .1       0   104.7      .1       0  111.65      .1       0
Bank Sta=104.7,111.65
XS Rating Curve= 0 ,0
Exp/Cntr=0.3,0.1

Type RM Length L Ch R = 1 ,2559.804,93.39,91.09,86.73
XS GIS Cut Line= 2
     617898.5416    4332261.2503     618050.9419    4332412.0631
#Sta/Elev= 30
       0  584.01    6.13  578.51    9.19   577.6   12.25  575.73   21.44  569.17
   27.57  564.09   30.63     562   45.94  555.19   49.01  554.41   55.13  550.22
   70.45  541.53   76.57  538.46   79.64   537.6    82.7  537.43   88.83  537.12
   91.89  537.74  101.08  540.27   107.2  542.44  110.27   543.7  119.46  548.66
  125.58  549.79  137.83  553.79  143.96  556.23  153.15  560.45  156.21  562.44
  162.34  563.95  192.97  579.84  199.09  580.34  205.22  582.38  214.41  584.45
#Mann= 3 , 0 , 0
       0      .1       0    82.7      .1       0   91.89      .1       0
Bank Sta=82.7,91.89
XS Rating Curve= 0 ,0
Exp/Cntr=0.3,0.1

Type RM Length L Ch R = 1 ,2468.713,89.4,91.29,92.69
XS GIS Cut Line= 2
      617832.766    4332377.2439     618007.1576    4332426.0144
#Sta/Elev= 30
       0  575.41   12.28  571.42   15.35  570.07   33.76  566.34    39.9  564.41
   42.97  563.12   52.18  558.66   58.31  553.31   70.59  546.54   73.66  544.15
   76.73  541.35   82.87  537.91   85.94  536.66   89.31  536.13   95.15  535.87
   98.21  535.97  104.35  537.61  113.56  539.48  122.77  542.56  128.91  545.33
  131.98  546.91  135.04  549.44  138.11  551.59  153.46  559.23  156.53  561.23
   159.6  563.69  171.88  569.86  174.94  571.66  178.01  574.78  181.08  576.52
#Mann= 3 , 0 , 0
       0      .1       0   89.31      .1       0   98.21      .1       0
Bank Sta=89.31,98.21
XS Rating Curve= 0 ,0
Exp/Cntr=0.3,0.1

Type RM Length L Ch R = 1 ,2377.421,72.98,91.42,102.24
XS GIS Cut Line= 4
     617817.6848    4332375.6564     617860.7398    4332462.0024
     617881.7921    4332482.3931     617943.0975    4332520.1192
#Sta/Elev= 30
       0  576.41   18.09  566.43   21.11  565.13   24.12  565.15   51.26  553.89
   54.27  553.97   57.29   553.1   75.38  544.82   84.42  539.74   90.45  538.83
   96.49   537.5     117  535.82  122.86  535.89  128.79  534.65  131.79   533.8
  134.83  533.87  137.79  534.99  143.79  537.96  146.79  538.89  149.79  540.24
  152.79  542.37  158.79  547.78  161.79  551.01  164.78  555.12  167.78  555.89
  170.78  557.56  182.78  566.53  185.78  569.66  188.78  571.54  197.78  575.91
#Mann= 3 , 0 , 0
       0      .1       0  128.79      .1       0  134.83      .1       0
Bank Sta=128.79,134.83
XS Rating Curve= 0 ,0
Exp/Cntr=0.3,0.1

Type RM Length L Ch R = 1 ,2286    ,102.94,91.47,81.3
XS GIS Cut Line= 4
     617808.1598    4332388.3564     617814.4771    4332466.9258
     617792.8619    4332525.5956      617801.016    4332564.5693
#Sta/Elev= 30
       0  567.18    9.09  562.05   12.13  562.04   27.28  553.88   33.35  550.86
   39.41  548.23   42.44  548.06   45.47  546.97   60.63  540.52    66.7  537.79
   69.73  537.38   75.79  535.48   99.66  531.54  105.62  530.84   108.6  530.39
  111.57  530.21  114.48  530.47  117.53   531.2  120.51   532.4  123.48  534.26
  135.39  543.82  138.37  543.88  141.35  545.55  144.41  548.09  147.47  550.27
  159.73  558.62  162.79  560.33  165.85  561.19  168.91  561.82  181.17  565.88
#Mann= 3 , 0 , 0
       0      .1       0  105.62      .1       0  114.48      .1       0
Bank Sta=105.62,114.48
XS Rating Curve= 0 ,0
Exp/Cntr=0.3,0.1

Type RM Length L Ch R = 1 ,2194.526,93.64,91.41,91.58
XS GIS Cut Line= 3
     617656.5532    4332479.6378     617752.3285    4332519.9618
      617791.491    4332592.3506
#Sta/Elev= 30
       0  568.08    3.06  566.37   15.28  557.94   21.39  551.58   30.56  545.11
   36.68  542.04   39.73  539.47   45.85  536.24   61.13   528.6   64.18  527.52
   67.24  526.71    70.3  526.41   73.35  526.53   76.41  526.98   82.52  528.71
   91.69  531.74  100.86  534.05  103.92  535.22  106.97  536.14  113.06  537.39
  122.21  540.62   128.3  542.42  131.35  543.84   134.4  545.54  137.45  546.84
  143.55  548.61  167.93  559.23  174.03  562.98  177.08  563.65  186.22   566.8
#Mann= 3 , 0 , 0
       0      .1       0   67.24      .1       0   76.41      .1       0
Bank Sta=67.24,76.41
XS Rating Curve= 0 ,0
Exp/Cntr=0.3,0.1

Type RM Length L Ch R = 1 ,2103.12 ,49.2,49.2,49.2
XS GIS Cut Line= 3
     617621.7869    4332566.3155     617693.6359    4332595.5961
      617778.493    4332601.1605
#Sta/Elev= 30
       0  558.05    2.98  556.03    5.97  554.39    8.95   553.1   14.92  551.45
    17.9  550.41   20.89  549.05   23.87  546.97   26.86  545.55   38.79  540.61
   41.78  539.17   44.76  537.27   59.68  530.83   62.67  529.16   65.65  528.08
   71.62  527.75   83.66  527.44   89.73  526.91   95.81   525.5   98.85  525.06
  101.88  525.36  104.92  527.18  120.11  531.56  123.14  532.66  126.18  535.31
  141.37  544.75   144.4  548.04  147.44  550.37  153.51  553.85  162.63   558.3
#Mann= 3 , 0 , 0
       0      .1       0   95.81      .1       0  101.88      .1       0
Bank Sta=95.81,101.88
XS Rating Curve= 0 ,0
Exp/Cntr=0.3,0.1

Type RM Length L Ch R = 1 ,2054    ,42.2,42.2,42.2
XS GIS Cut Line= 4
617619.8651778644332579.67319527617681.4219074594332633.13035518
617721.9197558774332656.88909292617814.2548502684332658.50900686
#Sta/Elev= 30
       0 553.237   3.846 550.076  14.453 543.622  24.204 538.712  29.708 535.331
  31.357 534.512  34.066 534.658  36.045  534.14  42.783 530.799  50.111 527.572
  52.706  527.02  55.858 526.765   84.27 525.327  88.376  524.61  93.256 523.098
  95.502 522.484  97.749  522.42 101.573 522.751 111.227 523.085 119.799  523.78
 128.481 525.828 140.006 526.763 144.684 527.483 158.454 528.824 162.685  529.57
 177.793 531.044 183.052 532.143 189.202 532.849 201.501  535.26 220.831 537.414
#Mann= 3 , 0 , 0
       0      .1       0  93.256      .1       0 101.573      .1       0
Bank Sta=93.256,101.573
XS Rating Curve= 0 ,0
Exp/Cntr(USF)=0,0
Exp/Cntr=0.3,0.1

Type RM Length L Ch R = 1 ,2011.762,105.42,91.52,80.94
XS GIS Cut Line= 3
     617597.1806    4332588.5406     617688.3047    4332694.2456
     617740.0559    4332726.6533
#Sta/Elev= 30
       0  557.85    3.03  555.62    6.07  552.83    18.2  545.04   24.27  542.69
   30.34   538.2   33.37  535.39   42.47  528.37   48.54  524.98   54.61  523.51
   57.64  523.25   72.81  523.66   84.95  523.19   91.02  521.76   94.05   521.6
   97.09   520.8  100.12  519.98  103.15  519.89  106.19  520.27  121.36  523.72
  130.46  526.24  136.53  528.54  142.61  531.76  157.88  537.09  160.93  538.39
  163.98  540.42   182.3  547.47  185.36  549.98  191.46  552.85  200.62  558.35
#Mann= 3 , 0 , 0
       0      .1       0   97.09      .1       0  106.19      .1       0
Bank Sta=97.09,106.19
XS Rating Curve= 0 ,0
Exp/Cntr=0.3,0.1

Type RM Length L Ch R = 1 ,1920.24 ,78.96,91.44,97.97
XS GIS Cut Line= 5
     617539.2367    4332746.4971     617593.7921    4332747.7069
     617618.2713    4332735.1613     617637.5214     4332717.855
     617737.6746    4332733.0034
#Sta/Elev= 30
       0  557.06    3.03  553.86    9.09  548.78   15.16  543.37   18.19  541.03
   21.22  539.27   33.35   530.9   36.38  529.43   42.44  527.54   45.47  526.95
   51.54  526.29   57.63  524.64   60.68  523.44   63.74  521.69   66.79  519.52
   72.91  518.04   79.02  516.95   87.83  517.95   114.1   519.7  120.24  521.28
  132.52  523.04  141.73  526.35     154  529.62  166.28  533.96  172.42  536.49
  178.56  540.74  193.91  547.56  196.98  549.73  200.05  552.38  209.25   558.1
#Mann= 3 , 0 , 0
       0      .1       0   72.91      .1       0   87.83      .1       0
Bank Sta=72.91,87.83
XS Rating Curve= 0 ,0
Exp/Cntr=0.3,0.1

Type RM Length L Ch R = 1 ,1828.8  ,77.76,90.94,94.72
XS GIS Cut Line= 5
     617521.6331    4332757.5038     617614.8206    4332811.2019
      617637.899    4332814.4813     617646.3383    4332817.2117
     617712.1334    4332847.4623
#Sta/Elev= 30
       0  557.51    6.15   555.2   15.36  551.31   18.44  549.34   21.51  546.15
   27.66     542    33.8  538.26   39.95  534.95   46.09  531.08   58.39  527.31
   61.46  526.46    67.6  525.24   82.97  523.04   89.11  521.74   95.26  520.97
  110.47  519.46  127.95  518.92  142.75  517.61  145.77     517  148.78  517.02
   151.8  518.51  157.84  523.05  166.89  528.56  169.91  531.42  172.92  533.98
  178.96   537.7  188.01  542.45  191.03  545.81  194.04  548.05  212.15  560.16
#Mann= 3 , 0 , 0
       0      .1       0  142.75      .1       0  148.78      .1       0
Bank Sta=142.75,148.78
XS Rating Curve= 0 ,0
Exp/Cntr=0.3,0.1

Type RM Length L Ch R = 1 ,1737.855,84.18,91.93,97.68
XS GIS Cut Line= 2
     617517.3997    4332762.7955     617621.1166    4332940.5959
#Sta/Elev= 30
       0  556.93    3.07   555.4    9.22  553.37   24.58  546.97   30.72  543.93
   36.87  540.36   39.94  539.64   52.23  532.61   67.59  524.98   76.81   522.8
   98.31  519.17  125.96  515.68  135.18  515.03  141.32  514.27  147.47  513.64
  150.54  513.79  153.61  514.64  156.68  516.39  159.76  519.03  162.83  522.25
   165.9     524  168.97  526.53  172.05  531.02  175.12  534.35  178.19  536.88
  193.55  548.87  196.62  550.98   199.7  551.52  202.77  553.91  205.84  556.88
#Mann= 3 , 0 , 0
       0      .1       0  141.32      .1       0  150.54      .1       0
Bank Sta=141.32,150.54
XS Rating Curve= 0 ,0
Exp/Cntr=0.3,0.1

Type RM Length L Ch R = 1 ,1645.92 ,95.45,90.2,61.81
XS GIS Cut Line= 5
      617474.008    4332798.7789     617508.4455    4332884.5255
      617498.307    4332908.5377     617500.8246     4332931.614
     617553.3831    4333001.9793
#Sta/Elev= 30
       0  556.23    2.98  554.72    5.96  553.77   29.81     539   32.79  537.61
   35.77  536.96   44.71   531.2   47.69  528.71   59.62  520.78    62.6  519.47
   68.56  518.63   89.42  514.39    95.3   512.6    98.2  512.12  101.09  510.71
  103.99   510.4  109.78   510.9  118.47  511.49  162.88  512.79  165.91  513.21
  168.94  514.69  171.97  517.79     175  520.09  178.02  521.95  193.17  530.96
   196.2  531.85  202.25  537.26  211.34  543.46  226.48  554.78  229.51  556.73
#Mann= 3 , 0 , 0
       0      .1       0  101.09      .1       0  109.78      .1       0
Bank Sta=101.09,109.78
XS Rating Curve= 0 ,0
Exp/Cntr=0.3,0.1

Type RM Length L Ch R = 1 ,1555.715,95.46,92.73,76.18
XS GIS Cut Line= 2
     617371.3494     4332862.279     617530.6995    4333032.5299
#Sta/Elev= 30
       0  548.93    6.14  544.53   15.34  535.92   18.41  534.77   24.55  529.45
   30.68  524.62   33.75  522.27   36.82  520.28   49.09  515.51   55.23  514.38
   61.37  511.92   64.43  510.33    67.5  509.04   70.57  508.59   73.64   509.1
   79.78  510.45   85.91  511.06  168.76  512.88  171.82  512.98  174.89  513.41
  177.96  515.32  181.03  518.07  187.17  521.93  196.37  527.25  199.44  528.39
  202.51  530.05  205.58  532.71  227.05  545.22  230.12  547.68  233.19  550.57
#Mann= 3 , 0 , 0
       0      .1       0    67.5      .1       0   73.64      .1       0
Bank Sta=67.5,73.64
XS Rating Curve= 0 ,0
Exp/Cntr=0.3,0.1
